HEC-RAS study R3.prj: San Jacinto Stage III Reach 3

--- R3.g29 (geometry) --- (continued)

Type RM Length L Ch R = 1 ,75818   ,500.841,500,500.043
XS GIS Cut Line= 6
    6277400.9622    2219887.2207    6276802.7563    2220412.7941
    6268628.6081    2227635.9124    6267610.4083    2228535.6485
     6267584.743    2228558.3279    6266588.6342    2229438.5433
#Sta/Elev= 30
       01424.796 338.115    1420 853.0611419.8051071.8451416.5881291.8641418.036
1318.554 1414.631345.2441414.8441425.313    14231452.002    1418 1638.831420.308
1798.968 1416.732015.9051416.0547363.7611413.8227483.864    14127497.2091411.134
7543.1891398.3517577.2781411.5217672.6071411.5217683.3551407.9647694.1041411.521
7734.1381410.2277840.8961413.4998973.8781413.4069170.2021415.73611657.52  1415.5
13051.381420.93413141.991420.625 13172.2    1418 13202.4    142214543.691429.159
#Mann= 3 ,-1 , 0
       0    .035       07483.864     .07       07577.278    .035       0
#XS Ineff= 3 ,-1
       0    2135    1428    2135    5563  1415.3    9418   14000  1415.4
Permanent Ineff=
       T       T       T
Bank Sta=7363.761,7840.896
XS Rating Curve= 0 ,0
Exp/Cntr=0.3,0.1

Type RM Length L Ch R = 1 ,75318   ,500.841,500,500.043
XS GIS Cut Line= 6
6277243.476495732219356.10864324    6276196.6814    2220281.1131
    6275931.9347    2220515.0577    6275854.2341     2220583.718
    6275507.9727    2220889.6934    6266443.7792    2228899.3036
#Sta/Elev= 30
       01423.989 595.4321419.0991243.8461418.0321297.2251429.2981350.604 1432.28
1492.2581429.8821577.4661420.5011630.846    14181743.1751420.0491790.9841417.958
1857.708    14221884.3971417.4951911.0871416.3757584.9661413.893 7678.21    1410
7742.7771410.0917782.8121398.0747811.6711409.4387844.331    14107972.4471413.753
12266.981417.131 12943.81420.13513140.121423.92413236.261421.56313454.671421.781
 13725.11423.985 13761.61426.02413814.98    142413955.621424.17314452.351427.563
#Mann= 3 ,-1 , 0
       0    .035       07742.777     .07       07844.331    .035       0
#XS Ineff= 3 ,-1
       0    1670    1428    1670 6017.18  1415.3 8872.18   12000  1415.4
Permanent Ineff=
       T       T       T
Bank Sta=7584.966,7972.447
XS Rating Curve= 0 ,0
Exp/Cntr=0.3,0.1

Type RM Length L Ch R = 1 ,74818   ,270,550,790
XS GIS Cut Line= 2
     6276530.736     2219318.683      6266298.93     2228360.059
#Sta/Elev= 30
       01422.031 266.0161420.281 292.7061423.641  332.741441.297 346.0851444.547
 439.4991448.094 572.947 1445.76 612.9821435.544 666.3611426.467 733.0851419.301
 787.8691417.753 985.4911422.3051040.016    14221080.051 1418.26 1155.521420.482
1424.7321416.4716468.9271412.3817078.1981413.8367221.266    14107232.0171409.644
7248.2271404.3887262.3961404.3817281.6731397.8517312.085    14107445.5341413.825
11448.981416.281 12316.4    142212609.98    142012632.481422.37113654.171426.953
#Mann= 3 ,-1 , 0
       0    .035       07221.266     .07       07312.085    .035       0
#XS Ineff= 3 ,-1
       0    1670    1428    1670    6324  1415.3    8178   13000  1415.4
Permanent Ineff=
       T       T       T
Bank Sta=7078.198,7445.534
XS Rating Curve= 0 ,0
Exp/Cntr=0.3,0.1

Type RM Length L Ch R = 1 ,74268   ,122,271,370
XS GIS Cut Line= 2
     6276213.599     2219458.017     6266340.809     2227116.229
#Sta/Elev= 30
       01449.993 142.002    1448 188.5681433.089 230.5931424.726  268.561420.084
 331.839    1418 382.4631418.149 546.988    1426 584.9551418.024 711.5131417.219
1597.4191420.2191880.155    14201961.7331416.0512124.8891415.5945368.848 1415.75
6383.251    14126774.8251413.5086921.665    14106938.0861404.356 6952.341404.745
6973.722 1397.68 6980.851398.7227001.4461408.4727014.103    14107084.8211413.807
9684.4771414.53110135.83    141810178.05    141610962.711415.64612494.811426.023
#Mann= 3 ,-1 , 0
       0    .035       06921.665     .07       07014.103    .035       0
#XS Ineff= 3 ,-1
       0    1706    1422    1706 6593.72  1415.3 7353.72   12000  1415.4
Permanent Ineff=
       T       T       T
Bank Sta=6774.825,7084.821
XS Rating Curve= 0 ,0
Exp/Cntr=0.3,0.1

Type RM Length L Ch R = 1 ,73997   ,79,79,79
BEGIN DESCRIPTION:
Cut Upstream of BNSF Railroad
jcc  14 DEC 2009
END DESCRIPTION:
XS GIS Cut Line= 2
     6276265.564     2219315.089     6266341.885     2226595.725
#Sta/Elev= 30
       01424.109  21.0791424.641  91.9891447.273 104.3911429.949 116.794    1424
 178.0061424.162  191.211427.173 216.0151422.305 302.8341421.729 501.277    1426
 600.498    14182839.7651414.3735469.3111415.7686963.0661412.7297075.298 1409.01
7092.2031401.4747110.7171397.4347136.7031402.0427146.487 1409.717167.9491412.453
7227.4441415.6377295.0641412.1789555.2231413.37810423.411415.84410490.13    1418
10820.291414.65910859.431419.18910882.311416.91711155.171416.72912308.01    1424
#Mann= 3 ,-1 , 0
       0    .035       07075.298     .07       07146.487    .035       0
#XS Ineff= 3 ,-1
       0    1979    1422    1979  7042.8  1415.3  7181.2   12000  1415.4
Permanent Ineff=
       T       T       T
Bank Sta=6963.066,7167.949
XS Rating Curve= 0 ,0
Exp/Cntr=0.5,0.3

Type RM Length L Ch R = 1 ,73918   ,136,136,136
BEGIN DESCRIPTION:
Copy of Section 73782
Upstream of Case Road Bridge and Downstream of BNSF Bridge
jcc  14 DEC 2009
END DESCRIPTION:
XS GIS Cut Line= 2
     6276155.702     2219298.933     6266032.209     2226726.123
#Sta/Elev= 30
       01421.269 391.276    1420 427.0311418.335 464.239    1420 898.3741419.992
 935.539    14182225.414    14182267.7511416.0812352.2781417.7692372.103 1416.28
2461.0641417.6652500.8751416.0852572.0451417.7292709.117    14165827.4981416.105
 6479.52    14126882.8691415.9696943.5261414.0826988.0281408.2347035.0151397.438
 7051.921401.7337065.1451407.9497115.2231414.0997310.4971412.7717565.9271414.064
8252.1881413.06210821.011416.00111763.05    142011819.181421.90812555.81    1426
#Mann= 3 ,-1 , 0
       0    .035       06988.028     .07       07065.145    .035       0
#XS Ineff= 3 ,-1
       0    2143    1422    2143    6972  1415.3    7096   14000  1415.4
Permanent Ineff=
       T       T       T
Bank Sta=6943.526,7115.223
XS Rating Curve= 0 ,0
Exp/Cntr=0.5,0.3

Type RM Length L Ch R = 3 ,73867   ,,,
BEGIN DESCRIPTION:
Case Road Bridge
This is based on field topo.  The sections are projected to the upstream and downstream sections.
jcc 6 August 2009
END DESCRIPTION:
Bridge Culvert--1,0,-1,-1, 0
Deck Dist Width WeirC Skew NumUp NumDn MinLoCord MaxHiCord MaxSubmerge Is_Ogee
59,23,3,0, 12, 12, 1415.3, , 0.98, 0, 5,5,,
     218     570     985    3272    5000  6979.1 6979.11  7090.8 7090.81    8000
   10160   11360
    1422    1418  1417.5  1415.3  1415.7  1416.7  1419.7  1419.7  1416.7  1415.4
  1416.1    1418
                                                  1414.7  1414.7
                
     218     570     985    3272    5000 6991.28 6991.28 7102.98 7102.98    8000
   10160   11360
    1422    1418  1417.5  1415.3  1415.7  1416.7  1419.7  1419.7  1416.7  1415.4
  1416.1    1418
                                                  1414.7  1414.7
                
Pier Skew, UpSta & Num, DnSta & Num=  ,7001.34, 2 ,7013.52, 2 , 0 , 0 , 0 ,,
    1.17    1.17
    1380    1420
    1.17    1.17
    1380    1420
Pier Skew, UpSta & Num, DnSta & Num=  ,7023.58, 2 ,7035.76, 2 , 0 , 0 , 0 ,,
    1.17    1.17
    1380    1420
    1.17    1.17
    1380    1420
Pier Skew, UpSta & Num, DnSta & Num=  ,7045.82, 2 ,7058, 2 , 0 , 0 , 0 ,,
    1.17    1.17
    1380    1420
    1.17    1.17
    1380    1420
Pier Skew, UpSta & Num, DnSta & Num=  ,7068.06, 2 ,7080.24, 2 , 0 , 0 , 0 ,,
    1.17    1.17
    1380    1420
    1.17    1.17
    1380    1420
BR Coef=-1 , 1 , 0 ,, 0 ,,,0.8,-1,2,0,
WSPro=,,,, 1 ,,,, 0 ,,,, 0 ,,,,-1 ,-1 ,-1 , 0 , 0 , 0 , 0 , 0
BC Design=,, 0 ,, 0 ,,,,,,
BC Use User HTab Curves=0
BC User HTab FreeFlow(D)= 0

Type RM Length L Ch R = 1 ,73782   ,618,409,265
BEGIN DESCRIPTION:
Cut Downstream of Case Road
END DESCRIPTION:
XS GIS Cut Line= 2
     6276076.022     2219188.714     6265951.617     2226616.616
#Sta/Elev= 30
       01437.383  30.5431425.602  55.349    1420 204.1811421.975 390.221    1418
 749.898 1417.09 824.3141419.527  898.731416.5931439.7621417.7771642.6241415.223
2322.4091417.3962994.7811414.3715859.7971414.3156145.058    14146182.2661411.998
6269.085    1414 6293.89 1410.296355.9031413.1936815.5921411.5676917.0231408.308
6984.644    14127008.2951408.575 7038.051397.2877062.8551407.1837079.835 1408.89
7102.979    14127286.104 1413.99  8439.1 1412.3111155.741416.18112556.961426.038
#Mann= 3 ,-1 , 0
       0    .035       07008.295     .07       07079.835    .035       0
#XS Ineff= 3 ,-1
       0    2143    1422    2143 6984.18  1415.3 7108.18   14000  1415.4
Permanent Ineff=
       T       F       F
Bank Sta=6984.644,7102.979
XS Rating Curve= 0 ,0
Exp/Cntr=0.5,0.3

Type RM Length L Ch R = 1 ,73373   ,900,556,295
XS GIS Cut Line= 2
     6275715.067     2218593.054     6265887.981     2226430.734
#Sta/Elev= 30
       01421.7421079.1411423.8191125.0051420.9821198.549  1398.51232.6331396.945
 1322.171398.3761386.125    14201424.4991418.7081475.6631398.4861663.642    1398
1744.274    14242511.7351414.9413171.1861417.9583315.5261410.6254174.5661410.844
4264.1041412.1794289.6861417.9926438.5761413.0316940.0461413.9757004.197    1420
7031.0931415.8257073.7881410.2267103.7081409.253 7137.831397.3697180.5241408.182
7231.6191410.0687287.2611417.7328269.2371410.789 11767.41418.39212569.841426.022
#Mann= 3 ,-1 , 0
       0    .035       07073.788     .07       07231.619    .035       0
#XS Ineff= 3 ,-1
       0    2382    1422    2382    6806  1415.3    7537   12000  1415.4
Permanent Ineff=
       T       F       F
#Block Obstruct= 3 ,-1
       0 1817.49    1422 3190.38 4294.24    1418
Bank Sta=7031.093,7287.261
XS Rating Curve= 0 ,0
Exp/Cntr=0.3,0.1

Type RM Length L Ch R = 1 ,72817   ,500.397,500,500.121
XS GIS Cut Line= 6
    6275857.4419    2217044.5198    6273400.7516    2219296.0591
    6269761.1881    2222631.5016    6269754.4644    2222637.6633
    6269661.5136    2222722.84736265848.183051432226217.53663142
#Sta/Elev= 30
       01425.725 363.893    1422 467.4961426.646  617.121420.634 1266.72    1422
 1934.331416.0012002.184    14162083.572    14242628.362    14242687.5641419.516
2776.3661404.4562870.313  1402.52965.265    14243013.1741417.933 3167.541416.007
 5000.941417.996 7197.291413.125 8078.961413.9468133.2171419.9848160.3451416.627
 8241.731408.7168275.2811397.228 8310.671408.0168336.6791408.9298418.0641417.261
8495.992    14208536.6851414.2428732.7141413.40610666.261413.406 13627.61425.996
#Mann= 3 ,-1 , 0
       0    .035       0 8241.73     .07       08336.679    .035       0
#XS Ineff= 3 ,-1
       0    3079    1424    3079    7555  1415.3    902313056.47  1415.4
Permanent Ineff=
       T       F       F
#Block Obstruct= 2 ,-1
 2146.26  2479.3 1424.04 2627.31 2960.35 1424.04
Bank Sta=8160.345,8418.064
XS Rating Curve= 0 ,0
Exp/Cntr=0.3,0.1

Type RM Length L Ch R = 1 ,72317   ,500.397,500,500.121
XS GIS Cut Line= 6
    6275128.8969    2217034.1096    6269419.8493    2222266.1105
    6269310.9003    2222365.9556    6266817.9029    2224650.6387
    6266528.6258     2224915.744     6265849.151    2225538.4419
#Sta/Elev= 30
       01426.473 389.9711420.0541191.7421418.2831827.771    1420  1854.91426.019
1889.0061415.3871936.285    14121963.4131414.0072004.105    14262037.0151418.179
2194.004    14182244.2281421.7362302.517    1408 2438.371406.0012543.5991406.832
2599.449    14222629.052    14183058.2781416.0094235.1891417.7426790.2711412.404
7631.761 1416.697687.4861409.702 7717.461408.7457750.1681396.5197782.4351408.045
7838.9741409.8187883.3761416.2667974.8531418.8149198.0641412.026 12646.41424.004
#Mann= 3 ,-1 , 0
       0    .035       07687.486     .07       07838.974    .035       0
#XS Ineff= 3 ,-1
       0    2637    1426    2637    6692  1415.3    882612587.19  1415.4
Permanent Ineff=
       T       F       F
#Block Obstruct= 2 ,-1
 1837.89 2010.57 1425.99 2220.26 2602.64 1421.99
Bank Sta=7631.761,7883.376
XS Rating Curve= 0 ,0
Exp/Cntr=0.3,0.1

Type RM Length L Ch R = 1 ,71817   ,500.397,500.004,500.121
BEGIN DESCRIPTION:
Blocked obstruction is EMWD WWTP.
jcc  20 AUG 2009
END DESCRIPTION:
XS GIS Cut Line= 6
     6274897.156    2216568.2786     6268837.788    2222121.3272
     6266479.211    2224282.8219    6265509.8915    2225171.1454
    6265500.7718    2225179.5029    6265487.3615    2225191.7927
#Sta/Elev= 30
       01425.185 136.3271420.4231024.382 1418.972030.844    14182273.027    1422
2356.4641407.4592652.483  1406.12688.0491407.2362741.288    14222788.465    1418
 3575.97    14164556.585 1417.075213.0411414.0087522.3541412.281  7706.21414.007
7734.5111419.7367758.798    14207784.0551415.2537807.2021410.1577862.4051408.964
7892.0071396.3127902.1511397.6117925.6111407.864 7951.211408.983  7997.1 1410.01
8017.6221413.7988123.2981416.0238287.502    14129761.1011413.12512832.071426.044
#Mann= 3 ,-1 , 0
       0    .035       07862.405     .07       0 7951.21    .035       0
#XS Ineff= 4 ,-1
       0    2777    1422    2777    6503  1415.3    930312763.59  1415.4
Permanent Ineff=
       T       F       F       F
#Block Obstruct= 1 ,-1
  2269.6 2725.99 1422.04
Bank Sta=7784.055,8017.622
XS Rating Curve= 0 ,0
Exp/Cntr=0.3,0.1

Type RM Length L Ch R = 1 ,71317   ,495.606,499.985,508.776
XS GIS Cut Line= 6
    6274714.5628    2216057.4067    6274442.6697    2216306.5805
    6274417.9132    2216329.2682    6269825.6327    2220537.8189
    6269666.6179    2220683.5463    6265124.4031    2224846.2147
#Sta/Elev= 30
       01423.522 194.1941420.735 356.9641422.039 370.5281424.041 448.4371420.906
1957.8191419.3432772.181    14162979.3931419.8343097.3431417.7217390.0661412.406
7922.8991413.9937939.3261418.1627967.3021419.932 7995.171414.6668026.5051408.107
8074.9671408.0318108.4151396.447 8115.661396.8628136.7271406.7398144.913    1408
8200.4271408.1448228.7371413.5678358.967    14168372.9751415.591 8388.261412.025
9749.9441412.028 10726.81415.12512713.061427.77513052.16    142813088.781431.214
#Mann= 3 ,-1 , 0
       0    .035       08074.967     .07       08144.913    .035       0
#XS Ineff= 3 ,-1
       0    2862    1424    2862    6379  1415.3    9847   14000  1415.4
Permanent Ineff=
       T       F       F
Bank Sta=7995.17,8228.737
XS Rating Curve= 0 ,0
Exp/Cntr=0.3,0.1

Type RM Length L Ch R = 1 ,70817   ,500.661,500.005,500.027
XS GIS Cut Line= 6
    6274105.4658    2216057.4067    6273559.9997    2216545.8269
    6271992.4237    2217949.4632    6271991.0083    2217950.7307
    6271758.6536    2218158.7852    6264680.1111     2224497.042
#Sta/Elev= 30
       0 1423.33  166.54    14202537.9071418.2812822.732    14163000.6041417.986
 3106.18    14165110.9871413.7136548.5971414.3516765.307    14146810.279    1412
7441.8151412.5357482.0841413.9817495.507 1417.81 7530.271417.5367576.0451408.688
7629.7371408.1157664.7531395.7197696.8531408.0587745.4251408.3047790.813 1416.32
7875.6871418.0287902.5331413.5917994.183    14128828.722    14128922.6831414.096
9343.3541413.5429405.911    14169473.026    141410137.861415.04812696.27 1432.07
#Mann= 3 ,-1 , 0
       0    .035       07629.737     .07       07696.853    .035       0
#XS Ineff= 3 ,-1
       0    2304    1422    2304    5613  1415.3    9748   12000  1415.4
Permanent Ineff=
       T       F       F
Bank Sta=7530.27,7790.813
XS Rating Curve= 0 ,0
Exp/Cntr=0.3,0.1

Type RM Length L Ch R = 1 ,70317   ,500.661,500,500.027
XS GIS Cut Line= 6
    6273413.7322    2216005.6467    6269080.6305    2219885.5853
    6268048.6346    2220809.6535    6268046.1537    2220811.8748
    6265310.5989    2223261.3407    6264531.8918    2223958.6094
#Sta/Elev= 30
       0    1424 231.9661420.5952915.3151414.0613023.3151416.2254862.2691415.918
5573.6881413.2295989.802    14166191.1471412.2166528.0931413.2376737.9641410.235
7063.6441413.7967093.9161408.2037157.6521408.1537187.6871395.7387197.8741396.638
 7224.721407.9827264.9891408.108 7305.151414.0967322.6041417.7577397.959    1418
7417.7471413.8347528.9141411.6387780.168    14147860.7061410.0878838.9281412.603
10998.881424.01611355.521428.866 11592.31428.21811713.11    143211967.481430.217
#Mann= 3 ,-1 , 0
       0    .035       07157.652     .07       0 7224.72    .035       0
#XS Ineff= 1 ,-1
       0    1706    1428
Permanent Ineff=
       T
Bank Sta=7063.644,7305.15
XS Rating Curve= 0 ,0
Exp/Cntr=0.3,0.1

Type RM Length L Ch R = 1 ,69817   ,500.661,500.002,500.027
XS GIS Cut Line= 6
    6272943.2486    2215755.7755    6270994.7448    2217500.5014
    6270193.8444    2218217.6423    6270085.1804    2218314.9422
    6269209.1478    2219099.3577    6264575.4207    2223248.4819
#Sta/Elev= 30
       01421.401  82.4771423.413 156.8191420.531 531.5891421.938 546.579    1420
 891.3671417.9312526.0141415.9062606.5521414.0392674.4251416.3793169.9661416.122
3214.938    14103255.1341408.5973349.8551417.781 3836.391411.9694129.375    1412
4474.1631415.8066258.066    14126566.3431403.693 6687.151406.0246752.7611410.385
6901.918    14126909.3551410.1816923.5191408.0616977.623    14087009.3021395.191
7049.5711407.994 7086.611408.0897127.5311411.6688997.1711414.00711299.281427.979
#Mann= 3 ,-1 , 0
       0    .035       06977.623     .07       07049.571    .035       0
#XS Ineff= 2 ,-1
       0    2113    1428    2113    4298 1415.85
Permanent Ineff=
       T       F
Bank Sta=6909.355,7127.531
XS Rating Curve= 0 ,0
Exp/Cntr=0.3,0.1

Type RM Length L Ch R = 1 ,69317   ,500.661,500,500.027
XS GIS Cut Line= 6
    6272405.3835    2215566.2388    6270968.3818    2216852.9566
    6270895.7975    2216917.9498    6267536.6199    2219925.8191
    6267261.3017    2220172.3439    6264476.1754    2222666.1971
#Sta/Elev= 30
       01419.858 408.043    1422 528.8511417.911 824.1571419.6742689.5661415.563
3173.185    14123469.0861415.9883499.0681409.771 3529.05    14083574.0221409.018
  3652.91416.6154193.3341412.0414623.3761414.4055562.4821411.1676394.709 1414.39
6555.7861412.0286582.631    1418 6616.211415.7556648.511 1410.116698.0841407.793
6705.1661407.5566737.0761394.9386770.5541407.7966832.639 1408.316871.9931416.913
6886.9841420.021 6943.131420.0816973.112    14128690.9321413.31310684.551426.078
#Mann= 3 ,-1 , 0
       0    .035       06698.084     .07       06770.554    .035       0
#XS Ineff= 2 ,-1
       0    2429    1428    2429    4087  1413.5
Permanent Ineff=
       T       T
Bank Sta=6616.21,6871.993
XS Rating Curve= 0 ,0
Exp/Cntr=0.3,0.1

Type RM Length L Ch R = 1 ,68817   ,587.366,581.311,564.226
XS GIS Cut Line= 6
    6271867.5185    2215376.7022    6268446.0672    2218440.3323
     6267313.766    2219454.2157    6267027.5635    2219710.4865
    6266914.9734    2219811.3019    6264250.8034    2222196.8485
#Sta/Elev= 30
       01421.783 800.0331416.0631041.7911419.8911068.6371414.7021140.0361413.483
 1309.721417.4322471.4191413.4843678.263    1418 3813.18    14083858.152    1408
3978.0781421.2033993.0691416.5394518.066 1411.97 4592.62    14164719.6981411.061
5243.1951412.663 5357.231417.226    60621408.2546236.4991417.8596271.667    1412
 6316.641417.9996343.8831416.0926424.4211407.805 6464.691394.8716491.5361405.896
 6558.631408.1066601.4641415.7196908.9581411.5948542.7931415.25110261.591429.979
#Mann= 3 ,-1 , 0
       0    .035       06424.421     .07       0 6558.63    .035       0
#XS Ineff= 2 ,-1
       0    2745    1428    2745    4392  1413.5
Permanent Ineff=
       T       T
Bank Sta=6343.883,6601.464
XS Rating Curve= 0 ,0
Exp/Cntr=0.3,0.1

Type RM Length L Ch R = 1 ,68236   ,440.603,418.742,376.128
XS GIS Cut Line= 6
    6271854.9762    2214400.7357    6270100.0362    2216040.1783
    6270021.4155    2216113.6248     6270009.351    2216124.8955
      6269725.97    2216390.2589    6263897.9128    2221847.7668
#Sta/Elev= 30
       01420.3321449.715    14181647.062    14221742.7751418.218 2509.17    1414
3704.1221417.8994892.967    14125020.8331415.8135057.3671412.0475211.025 1410.29
5313.4361415.7985413.5651414.0315518.2571418.4815619.0641413.7466030.062    1414
6125.961 1407.07 6358.861410.7066688.6671404.3656852.0581409.8186906.8571417.997
6920.5581417.9736937.379    14127006.5161415.988 7098.311406.474 7127.571394.347
7167.1561406.3517232.9121408.1597268.286 1414.388714.3411414.026 10965.91430.396
#Mann= 3 ,-1 , 0
       0    .035       0 7098.31     .07       07167.156    .035       0
#XS Ineff= 2 ,-1
       0    4150    1428    4150    5742  1413.5
Permanent Ineff=
       T       F
Bank Sta=7006.516,7268.286
XS Rating Curve= 0 ,0
Exp/Cntr=0.3,0.1

Type RM Length L Ch R = 1 ,67817   ,494.922,499.973,511.295
XS GIS Cut Line= 6
    6270845.6578    2214251.3503    6269675.7065    2215424.9974
    6269663.8418    2215437.6703    6267902.4543    2217319.0645
    6267847.6979    2217377.5514    6263748.7983    2221755.7168
#Sta/Elev= 30
       01419.9581323.335    14222239.896  1416.53185.0941416.8443682.677    1412
4882.4871417.4385208.5651407.9785643.343 1405.835787.8151408.468 5862.82    1414
6034.388    14146213.9841420.7886253.5651418.9866283.9511412.0956360.3031412.074
6376.852    14166425.4491413.5316506.6211406.0796538.6471394.3066566.9471405.983
6638.3081408.2546678.2191415.9896756.2331417.6566795.594    14126952.2591411.134
8185.6181414.9699941.4381426.61810038.991429.96910102.921427.21910384.191429.075
#Mann= 3 ,-1 , 0
       0    .035       06506.621     .07       06566.947    .035       0
#XS Ineff= 3 ,-1
       0    4170    1428    4170    5645  1413.5    7468   10329  1413.5
Permanent Ineff=
       T       T       T
Bank Sta=6425.449,6678.219
XS Rating Curve= 0 ,0
Exp/Cntr=0.3,0.1

Type RM Length L Ch R = 1 ,67317   ,250,250,250
XS GIS Cut Line= 2
     6269983.315     2214531.662     6263478.697     2221233.914
#Sta/Elev= 30
       0    1424 997.587 1420.461308.7491421.7381823.731    14162157.3721416.749
2486.7921413.888  3593.51416.4833678.554 1414.254224.181    14184674.9541415.846
4755.4481407.3224781.0321409.9844795.1761408.4544823.4631413.8774875.537    1416
 4942.111414.1745587.2241412.8355717.4741405.8915742.8051394.8395749.8761394.133
5778.1641404.8185795.2591406.013 5878.87 1411.76 7282.561416.0468072.2821421.181
8734.2011428.5649059.5071429.6819149.177    1432 9209.38    14309339.7131430.011
#Mann= 3 ,-1 , 0
       0    .035       05717.474     .07       05795.259    .035       0
#XS Ineff= 3 ,-1
       0    3843    1428    3843    5331  1413.5    6064 9339.97  1413.5
Permanent Ineff=
       T       T       T
Bank Sta=5587.224,5878.87
XS Rating Curve= 0 ,0
Exp/Cntr=0.3,0.1

Type RM Length L Ch R = 1 ,67067   ,220,220,220
BEGIN DESCRIPTION:
Section Taken Just Upstream of Goetz Road - This section will be skewed with Bridge  jcc 11 DEC 2009
END DESCRIPTION:
XS GIS Cut Line= 2
     6265803.439     2215602.343     6265778.971     2224145.867
#Sta/Elev= 30
       01424.016  62.2561423.898 161.2511420.089 239.033    1420  281.461418.011
 635.015 1417.88 685.0291416.0591320.9111413.8331384.5511412.0221773.461    1412
1844.1721413.6981917.9061412.539 1957.311411.5271985.5941406.5252013.8781404.271
2035.0921394.7792042.1631393.7692063.3761403.1622070.4481404.8172105.803    1410
2261.3671411.8623583.6621414.8913979.6441414.1834121.065  1415.94425.1221416.018
4460.4781417.4014580.6871416.0315160.5171421.1185818.128    14226041.208    1424
#Mann= 3 ,-1 , 0
       0    .035       02013.878     .07       02070.448    .035       0
#XS Ineff= 3 ,-1
       01214.102    14281214.1021986.093  1413.52086.9554242.641  1413.5
Permanent Ineff=
       T       T       T
Bank Sta=1917.906,2261.367
XS Rating Curve= 0 ,0
Skew Angle= 45
Exp/Cntr=0.5,0.3

Type RM Length L Ch R = 3 ,66966   ,,,
BEGIN DESCRIPTION:
Goetz Road Bridge
This is based on field topo.  The sections taken along the Goetz Road and then skewed 45 degrees to match the direction of flow.
END DESCRIPTION:
Bridge Culvert--1,0,-1,-1, 0
Deck Dist Width WeirC Skew NumUp NumDn MinLoCord MaxHiCord MaxSubmerge Is_Ogee
70,42,3,45, 15, 16, 1413.5, , 0.98, 0, 2,2,,
  72.125 436.285 648.417 947.5231269.9641529.4721821.5071986.0931986.0932086.955
2086.9552437.3974449.8234676.8044993.319
    1428    1424    1422    1420    1418    1416    1414  1413.5  1413.5  1413.5
  1413.5    1414    1416    1418    1420
                                                                 1412.25 1412.25
                                        
  50.205  364.16 622.254  921.361198.5461466.5391750.089 1814.04 1814.041914.902
1914.9022369.515 4381.944652.7635008.4375126.524
    1428    1424    1422    1420    1418    1416    1414  1413.5  1413.5  1413.5
  1413.5    1414    1416    1418    1420    1422
                                                                 1412.25 1412.25
                                                
Pier Skew, UpSta & Num, DnSta & Num=  ,2000.143, 2 ,1828.09, 2 , 0 , 0 , 0 ,,
     1.5     1.5
    1380    1415
     1.5     1.5
    1380    1415
Pier Skew, UpSta & Num, DnSta & Num=  ,2017.842, 2 ,1845.789, 2 , 0 , 0 , 0 ,,
     1.5     1.5
    1380    1415
     1.5     1.5
    1380    1415
Pier Skew, UpSta & Num, DnSta & Num=  ,2036.694, 2 ,1864.641, 2 , 0 , 0 , 0 ,,
     1.5     1.5
    1380    1415
     1.5     1.5
    1380    1415
Pier Skew, UpSta & Num, DnSta & Num=  ,2055.284, 2 ,1883.23, 2 , 0 , 0 , 0 ,,
     1.5     1.5
    1380    1415
     1.5     1.5
    1380    1415
Pier Skew, UpSta & Num, DnSta & Num=  ,2072.94, 2 ,1900.887, 2 , 0 , 0 , 0 ,,
     1.5     1.5
    1380    1415
     1.5     1.5
    1380    1415
Abutment Skew #Up #Dn= , 2 , 2
1986.0932017.842
 1411.25    1404
 1814.041845.789
 1411.25    1404
Abutment Skew #Up #Dn= , 2 , 2
2055.2842086.955
    1404 1411.25
 1883.231914.902
    1404 1411.25
BR Coef=-1 , 1 , 0 ,, 0 ,,,0.8,-1,1.2,0,
WSPro=,,,, 1 ,,,, 0 ,,,, 0 ,,,,-1 ,-1 ,-1 , 0 , 0 , 0 , 0 , 0
BC Design=,, 0 ,, 0 ,,,,,,
BC Use User HTab Curves=0
BC User HTab FreeFlow(D)= 0

Type RM Length L Ch R = 1 ,66847   ,30,30,30
BEGIN DESCRIPTION:
Section Taken Just Downstream of Goetz Road - This section will be skewed with Bridge  jcc 11 DEC 2009
END DESCRIPTION:
XS GIS Cut Line= 2
     6265647.533     2215702.258     6265623.687     2224029.063
#Sta/Elev= 30
       01431.627 387.5861429.022 437.0841428.018 458.2981424.478 479.5111423.966
 500.7241424.423 543.1511429.698 649.2171428.236 712.8571429.895 726.9991428.064
 809.8321427.719 833.0661420.647 882.5631414.4411483.5151410.0181716.3771411.978
1788.4451410.0051844.2321405.0551864.4461394.6341871.4971393.7811879.5881395.899
1899.7011406.2861927.9051409.9451951.5481410.3481985.6541409.0332692.764    1414
4375.685 1416.014616.103    14204672.6711418.6144693.8841420.1835887.9641423.928
#Mann= 3 ,-1 , 0
       0    .035       01844.232     .07       01899.701    .035       0
#XS Ineff= 3 ,-1
       01146.927    14281146.927 1814.04  1413.51914.9023535.534  1413.5
Permanent Ineff=
       T       F       F
Bank Sta=1788.445,1951.548
XS Rating Curve= 0 ,0
Skew Angle= 45
Exp/Cntr=0.5,0.3

Type RM Length L Ch R = 1 ,66817   ,488.943,490.173,495.119
XS GIS Cut Line= 2
     6268787.315     2214851.759      6263416.04     2220689.036
#Sta/Elev= 30
       01424.011 691.1921422.632 786.3171420.346 1370.661415.9311642.4471418.957
2083.9071417.0572415.9841422.7382471.399 1419.932586.3871418.0653154.402    1414
3697.5031416.6493759.9041417.7673775.9781419.7813939.0511414.8084380.175    1412
4468.7851412.006 4513.09    14144564.161 1410.154624.6141410.0624675.5421405.351
4695.3851395.7244705.0791393.7554734.6161405.991 4759.081409.9866876.027 1420.07
7200.4991424.1857335.1721427.979 7540.411430.0317673.5191428.025 7932.491431.996
#Mann= 3 ,-1 , 0
       0    .035       04675.542     .07       04734.616    .035       0
#XS Ineff= 3 ,-1
       0    3325    1428    3325    4590  1413.5    5063 7932.49  1413.5
Permanent Ineff=
       T       F       F
Bank Sta=4624.614,4759.08
XS Rating Curve= 0 ,0
Exp/Cntr=0.3,0.1

Type RM Length L Ch R = 1 ,66327   ,512.084,509.915,510.645
XS GIS Cut Line= 6
    6267944.6375    2215068.9381    6265311.6366    2217905.6875
      6265242.75    2217979.9049    6264399.7486      2218888.14
    6264393.0136     2218895.396    6263394.9866    2219970.6531
#Sta/Elev= 30
       01427.813 261.2061425.878 406.6491427.012 602.2991424.011 769.139    1418
1361.9051421.438 1977.681414.0422348.6941416.4442512.4191420.8663099.0981413.594
3187.5061414.0823229.9611416.4233344.685    14163378.5571412.0533606.1431410.146
3760.6591410.0763794.9281414.9673835.8591413.4793888.0271406.0743929.532    1406
3958.9311393.3753972.296 1395.79 3988.331403.6033999.583    14064047.128 1407.85
4081.4461413.231 4152.111413.9784206.9821410.027 4901.321414.0046717.493 1430.04
#Mann= 3 ,-1 , 0
       0    .035       03929.532     .07       03999.583    .035       0
#XS Ineff= 3 ,-1
       0    3068    1428    3068    3517  1413.5    4486 6687.76  1413.5
Permanent Ineff=
       T       F       F
Bank Sta=3835.859,4081.446
XS Rating Curve= 0 ,0
Exp/Cntr=0.3,0.1

Type RM Length L Ch R = 1 ,65817   ,510.902,499.882,492.717
XS GIS Cut Line= 6
    6265799.1095    2216622.3803    6265003.0642    2217487.4889
    6264943.4484    2217552.2767    6264628.0409    2217895.0485
    6264144.0191    2218421.0629    6263070.3566    2219587.8743
#Sta/Elev= 30
       0    1416  85.2341420.171 188.6121421.966 218.1491428.063 309.8451428.357
 533.9581427.914 649.5791425.857 867.0091414.1451016.492 1410.411122.2421410.156
1165.9751412.023 1192.86    14181220.3331416.2551270.8621406.3361315.458    1406
 1327.481404.4231348.7111394.5381355.7881393.0981384.0971404.9711396.9951406.123
1437.7631406.3041483.1781415.0631530.495    14161559.2081410.7691589.5681410.515
1912.5321413.8233067.0411420.2473671.9061426.294  3908.21425.486 4042.651427.953
#Mann= 3 ,-1 , 0
       0    .035       01315.458     .07       01396.995    .035       0
#XS Ineff= 2 , 0
       0     979    1428               0
Permanent Ineff=
       T       F
Bank Sta=1220.333,1483.178
XS Rating Curve= 0 ,0
Exp/Cntr=0.3,0.1

Type RM Length L Ch R = 1 ,65317   ,585.896,499.588,419.787
XS GIS Cut Line= 2
     6265337.133     2216337.679     6262691.738     2219366.285
#Sta/Elev= 30
       01428.007  16.872    1426  69.9821424.763 162.9251427.313 229.313 1426.14
 282.3841423.345 530.436  1424.1 721.7891421.538  753.57    1424 844.776    1424
 853.3611422.994 879.9161411.248 890.379    14101065.8031410.051 1097.411415.585
1132.8461415.0171189.5431406.3021225.1341406.1551238.412 1402.481253.3281395.149
1264.9671392.8531291.5221404.5061300.8061405.9811345.4611406.0681392.0121414.874
1437.6151415.7111451.7691412.0061501.3791411.3193018.5191421.0334021.265 1424.79
#Mann= 3 ,-1 , 0
       0    .035       01225.134     .07       01300.806    .035       0
Bank Sta=1132.846,1392.012
XS Rating Curve= 0 ,0
Exp/Cntr=0.3,0.1

Type RM Length L Ch R = 1 ,64817   ,549.221,499.439,451.105
XS GIS Cut Line= 3
     6264663.061     2215968.432     6263644.063     2217823.711
     6262655.654       2219382.4
#Sta/Elev= 30
       01426.153 104.911    1424 252.7281426.095 527.046    1426 585.0851425.034
  606.91    1422 663.9551421.994 675.364    1424 778.046    1424 812.273 1410.79
 820.1011410.123 960.0221409.972 994.8181411.8741017.6361414.682 1062.851413.509
1099.9441406.1671143.135    14061154.5451404.8581177.3631393.6441187.4841392.621
 1211.591403.9011222.9991406.0311269.3221407.0591306.1441412.8671314.271    1414
1359.908    14141374.4351411.9831473.9981411.2752657.4531419.074 3962.36 1425.18
#Mann= 3 ,-1 , 0
       0    .035       01143.135     .07       01222.999    .035       0
Bank Sta=1062.85,1306.144
XS Rating Curve= 0 ,0
Exp/Cntr=0.3,0.1

Type RM Length L Ch R = 1 ,64318   ,532.348,499.504,468.255
XS GIS Cut Line= 2
     6264072.036     2215703.426     6262650.272     2219318.767
#Sta/Elev= 30
       0    1428  29.0741427.998  93.443    1424 247.667    1424 298.9361425.697
 415.807 1426.01  598.481423.656 748.916    1426 759.6621424.758 781.1531418.268
 824.1351415.875 946.7841412.593 963.8261412.997 985.3461415.9981006.8081415.951
1028.2991414.1791071.2811406.8041114.2631405.8881125.0081405.0951146.4991394.366
1157.2451392.2991189.481 1405.951232.4631406.265 1286.191414.5031318.4271415.881
1347.833 1412.041372.1541411.5461554.8271411.0572682.0911419.9973884.8561425.528
#Mann= 3 ,-1 , 0
       0    .035       01114.263     .07       01189.481    .035       0
Bank Sta=1028.299,1286.19
XS Rating Curve= 0 ,0
Exp/Cntr=0.3,0.1

Type RM Length L Ch R = 1 ,63818   ,500.024,500,500.222
XS GIS Cut Line= 6
    6263571.6532    2215289.0961    6263217.3778    2216482.3522
    6262895.6989    2217565.8176    6262782.8345    2217945.9632
    6262578.2574    2218635.0111    6262421.0415    2219164.5396
#Sta/Elev= 30
       01427.629  11.7771429.842 108.1621429.992 220.406    1428 804.5661424.395
 877.5861425.993   981.9    14261002.7631417.3861013.1951416.0761190.529    1414
1207.751 1417.661221.8231418.0391247.9671415.835 1292.291406.9261336.5691405.997
1344.4881404.7091367.8631393.6691378.2951392.0441409.5891404.8241457.0951406.136
1505.3551414.5271513.904    14161536.102    14161544.8281414.4891553.555    1416
1584.849 1416.011605.712    14121668.3011411.3132019.566 1412.364082.2951427.948
#Mann= 3 ,-1 , 0
       0    .035       0 1292.29     .07       01457.095    .035       0
Bank Sta=1247.967,1505.355
XS Rating Curve= 0 ,0
Exp/Cntr=0.3,0.1

Type RM Length L Ch R = 1 ,63318   ,484.415,499.819,514.433
XS GIS Cut Line= 6
    6263049.1812    2215292.1281    6262735.8303    2216347.5437
    6262534.2464    2217026.5107    6262438.7653    2217348.1059
    6262417.2653    2217420.5217    6262111.5792    2218450.1211
#Sta/Elev= 30
       01428.143  19.0451429.844   50.34    1428 603.2061426.306 686.6571423.039
 728.3831425.732 801.403 1425.69 825.2851424.204 863.992    14141020.463    1412
1051.758    1416 1093.381414.6451124.7781411.3381145.6411406.6391187.3661405.101
1208.2291394.6791218.6611391.7561229.0921394.4311249.9551404.759 1257.071405.287
1302.112    14061348.1041413.3051402.7821413.9791434.9551411.2381535.6331410.454
1942.4591410.0942349.285  1419.22787.4051426.1112996.0341425.2163308.701    1428
#Mann= 3 ,-1 , 0
       0    .035       01187.366     .07       0 1257.07    .035       0
Bank Sta=1093.38,1348.104
XS Rating Curve= 0 ,0
Exp/Cntr=0.3,0.1

Type RM Length L Ch R = 1 ,62818   ,501.027,500.015,500.265
XS GIS Cut Line= 6
    6262665.1355     2215025.788    6262628.7483    2215132.1668
    6261844.0206    2217426.3413    6261696.8594    2217856.5717
    6261660.8127     2217961.955    6261592.5569    2218161.5032
#Sta/Elev= 30
       01424.164 110.5481425.848 195.0981422.618 311.3551426.134 660.1261424.001
  920.081424.844 967.3311424.043  987.761417.9761006.7061416.0651199.1361415.918
1241.4111413.6111283.6871405.9531315.393  1405.61325.9621405.5241357.6681391.558
1368.2371392.8991389.3751403.4641424.0871405.2281452.7881405.9471484.4941411.855
1760.398 1408.031976.5231412.0042800.5981420.0463075.3871425.7593107.0941427.855
  3138.81433.9713149.3691434.1283170.5061429.3223212.7821427.031 3330.221428.005
#Mann= 3 ,-1 , 0
       0    .035       01315.393     .07       01424.087    .035       0
Bank Sta=1241.411,1484.494
XS Rating Curve= 0 ,0
Exp/Cntr=0.3,0.1

Type RM Length L Ch R = 1 ,62318   ,441.519,498.258,545.036
XS GIS Cut Line= 6
    6262193.9493    2214858.4017    6261870.8543    2215802.9796
    6261774.1023    2216085.8366    6261709.8765    2216273.6029
    6261687.9728    2216337.6387    6261145.1096    2217924.7155
#Sta/Elev= 30
       01491.213  86.6871453.821 118.3541437.644 128.9231434.062 498.8321424.083
 741.9151424.476 794.7591423.863 811.693    1422 984.9971424.074 995.5661423.366
1016.7041416.5391058.9791414.7511145.4661412.0261196.374    1412 1228.08    1414
1291.4931412.6311336.5151404.3091354.9061402.1071376.0441391.7771381.7191391.592
1386.6131391.689 1407.751401.949 1428.97  1404.11492.301    14121567.6071411.974
1620.4511409.4541874.103    14102138.3231413.8792677.333 1418.013273.7631428.065
#Mann= 3 ,-1 , 0
       0    .035       01336.515     .07       0 1428.97    .035       0
Bank Sta=1291.493,1492.301
XS Rating Curve= 0 ,0
Exp/Cntr=0.3,0.1

Type RM Length L Ch R = 1 ,61820   ,427.551,498.528,543.781
XS GIS Cut Line= 2
     6261940.961      2214750.17     6260556.217     2217330.166
#Sta/Elev= 30
       01517.877  34.2931505.969  51.536 1502.75   79.691495.008 102.3891486.028
 125.088 1481.45 181.834 1460.58 243.5571439.699  261.281433.912 272.6291431.966
 613.1091425.998 669.8551422.026 794.6981421.961 828.7461423.893 959.9411425.725
1010.3351420.1291159.3471416.0161233.2011417.7841277.5141411.9231307.0551406.001
1350.8151404.2021373.5241393.6551384.8631391.0171417.8361403.9281458.1261410.239
1532.4041409.9821577.8011408.0212485.7471416.6252848.926 1423.822928.1221427.576
#Mann= 3 ,-1 , 0
       0    .035       01350.815     .07       01417.836    .035       0
Bank Sta=1277.514,1458.126
XS Rating Curve= 0 ,0
Exp/Cntr=0.3,0.1

Type RM Length L Ch R = 1 ,61321   ,389.412,499.567,583.656
XS GIS Cut Line= 6
    6261789.9075    2214604.2509    6260715.9898    2215865.9574
     6260675.789     2215913.188    6260481.8705    2216141.0156
     6260313.931    2216338.32176260046.317746252216652.73055002
#Sta/Elev= 30
       0 1528.85  86.8481517.746 151.9861513.691 270.6951499.721 365.0851456.915
 388.8831449.963 410.3841438.909  428.931432.469 968.065 1420.011073.1551419.919
1297.7761411.4511348.9931405.4161392.2641403.9421399.3581402.9431429.0951390.804
1441.5621394.2351463.2031404.0161491.5791409.7621597.9871406.2551647.6441412.111
1712.182 1427.621719.6341425.7651754.7681433.2881772.297    14341795.8871432.708
1875.3641420.9911974.6791416.982 2119.881418.881 2289.591417.4312760.2721423.085
#Mann= 3 ,-1 , 0
       0    .035       01392.264     .07       01463.203    .035       0
#XS Ineff= 2 , 0
                         1718.06         1434.46
Permanent Ineff=
       F       F
Bank Sta=1297.776,1491.579
XS Rating Curve= 0 ,0
Exp/Cntr=0.3,0.1

Type RM Length L Ch R = 1 ,60821   ,502.739,500.048,501.639
XS GIS Cut Line= 2
     6261785.927     2214562.971       6259432.2     2215927.567
#Sta/Elev= 30
       01533.526  63.0331519.441  86.1511512.686 114.4721500.969 132.388 1496.76
 167.0651498.045 247.9781489.863 305.7741485.675 381.9071476.966 469.7111463.871
 513.2261454.313 573.0391432.126 601.4161430.502 999.3181427.9881022.4361426.041
1045.5541419.8911257.3381412.1721288.2951406.0471350.609    1404 1391.651404.288
1428.2351409.9051545.3071410.0221611.9491412.0061958.7211433.0162085.8711437.818
2166.7841442.8862335.5411448.838 2386.761448.8392536.6741445.087 2720.691438.019
#Mann= 3 , 0 , 0
       0    .035       01257.338    .035       01428.235    .035       0
Bank Sta=1257.338,1428.235
XS Rating Curve= 0 ,0
Exp/Cntr=0.3,0.1

Type RM Length L Ch R = 6 ,60723   ,,,
Lateral Weir Pos= 3
Lateral Weir TW Multiple XS=0
Lateral Weir Coef=2
LW OverFlow Method 2D=False
Lateral Weir WSCriteria=-1
Lateral Weir Flap Gates= 0
Lateral Weir Hagers EQN= 0 ,,,,,
Lateral Weir SS=0.05,0.05,
Lateral Weir Type= 0
Lateral Weir Connection Pos and Dist= 3 ,
Lateral Weir SE= 0
Lateral Weir Centerline= 0
LW Div RC= 9 ,False,
 1393.27      50 1394.41     100 1396.18     200 1397.93     300 1402.82     400
 1406.12     500 1410.16     600 1414.94     700 1420.44     800

Type RM Length L Ch R = 1 ,60321   ,475.681,499.787,516.943
XS GIS Cut Line= 6
    6261531.2769    2214132.6535    6260617.4146    2214662.4741
    6260444.8318    2214762.5307    6260439.9567    2214765.3572
    6259635.9465    2215231.4899    6259315.6303    2215417.1965
#Sta/Elev= 30
       01443.241  80.776 1440.55 232.3971441.906  288.841440.022 311.9581436.023
 473.785    1434 496.9031431.941 620.1971428.698 653.4231425.345 797.4391426.781
1022.6311420.107 1111.991414.218 1155.771412.5371256.7751413.6581306.0381405.977
1363.833    14041410.069    14041425.0651405.9171444.7471408.5181479.4241409.982
1563.7321410.1791599.8361412.3981652.3281419.1611658.4761418.3021702.2081421.967
1815.3741420.0931977.2011427.7392147.1081424.8492293.4481427.6892573.3781430.424
#Mann= 3 ,-1 , 0
       0    .035       01306.038     .07       01425.065    .035       0
Bank Sta=1256.775,1479.424
XS Rating Curve= 0 ,0
Exp/Cntr=0.3,0.1

Type RM Length L Ch R = 1 ,59821   ,332.534,491.272,538.845
BEGIN DESCRIPTION:
Blocked Area is WQ Marsh for Adjacent Tract
jcc  20 Aug 2009
END DESCRIPTION:
XS GIS Cut Line= 3
     6260955.898     2213971.706     6260586.032     2214142.223
     6259846.974     2214513.309
#Sta/Elev= 30
       01428.132 137.096    1428 213.431 1429.11 258.2241427.917 280.2471425.836
  302.271416.635  311.411413.538 324.293    1412 386.7791412.494 390.3621413.063
 402.8921418.908 412.4681420.172 434.8471420.579 446.0371419.721 457.2271417.845
 498.7581416.094 557.9351415.224 692.2121411.909 736.9711410.036 915.9241405.998
 927.198 1404.38  938.04    1404 953.1711404.186 994.336    14081050.2851408.002
1072.6651409.2971083.8541410.3731128.6141420.3011184.1021423.5041234.2691428.373
#Mann= 3 , 0 , 0
       0    .035       0 915.924     .07       0 994.336    .035       0
#Block Obstruct= 1 ,-1
  294.87  426.78 1420.04
Bank Sta=915.924,994.336
XS Rating Curve= 0 ,0
Exp/Cntr=0.3,0.1

Type RM Length L Ch R = 1 ,59330   ,700.378,498.855,440.172
XS GIS Cut Line= 2
     6260454.991     2213867.925     6259649.991     2213949.983
#Sta/Elev= 30
       01420.783   3.6141420.162  13.6661418.822  23.7181417.844  73.9771416.031
 194.5991414.097 264.9611412.365 285.0651411.734 315.6711410.271 375.5311408.125
 395.6351407.858 455.946    1406 526.3091405.972 534.5991405.721 546.4121405.604
 556.4641404.805 566.5161402.828 576.5681402.968  586.621405.512 606.7231408.222
 616.7751409.251 626.8271410.517  646.931414.026 667.0341416.164 687.1381419.844
 707.2411424.092 737.3971429.833 767.5521435.828 787.6561439.276 809.1721444.014
#Mann= 3 , 0 , 0
       0    .035       0 546.412     .07       0  586.62    .035       0
Bank Sta=546.412,586.62
XS Rating Curve= 0 ,0
Exp/Cntr=0.3,0.1

Type RM Length L Ch R = 1 ,58831   ,624.909,491.981,412.339
XS GIS Cut Line= 2
     6260113.691     2213207.505     6259512.807     2213616.378
#Sta/Elev= 30
       0 1422.07  51.1581420.167  75.3491419.484 169.2751415.914 256.7821411.915
 291.637    1410 329.3551408.394 377.7371406.074 426.1191404.033 428.3941403.796
 431.7381403.149  442.791400.437 449.513    1400 450.3111400.071 457.1861402.298
 462.4061403.751 486.5971405.829 498.693    1406 510.7881404.886 522.884 1406.36
 547.0751408.151 565.1521409.882 579.5481411.655 595.4571413.891 615.5371416.098
 645.0461417.947 673.1191420.551 687.5141421.596  701.911422.449   726.81423.494
#Mann= 3 , 0 , 0
       0    .035       0 426.119     .07       0 462.406    .035       0
Bank Sta=426.119,462.406
XS Rating Curve= 0 ,0
Exp/Cntr=0.3,0.1

Type RM Length L Ch R = 1 ,58339   ,575.329,494.229,395.965
XS GIS Cut Line= 2
     6259434.833     2212951.526     6259164.833     2213589.526
#Sta/Elev= 30
       01415.866  42.1961414.006   96.491411.935 118.2071410.592 129.065 1410.01
 150.783    1410 154.3471409.928 161.6411409.981   172.51407.331 183.359 1405.85
 215.9341404.051 223.0151402.927 230.6451401.341 237.6521400.018  248.51    1400
 253.5341400.202 259.3691400.669 268.7931402.754 270.2271402.965 281.0861404.026
 335.3791405.764 346.2381406.033 389.6721407.704 422.2481409.746 465.6831412.019
 498.2591414.087 558.7231416.413 595.9861417.522 639.4211418.244  692.781419.654
#Mann= 3 , 0 , 0
       0    .035       0 215.934     .07       0 281.086    .035       0
Bank Sta=215.934,281.086
XS Rating Curve= 0 ,0
Exp/Cntr=0.3,0.1

Type RM Length L Ch R = 1 ,57845   ,514.213,499.263,481.295
XS GIS Cut Line= 2
     6258808.677     2212909.698     6258922.502     2213659.637
#Sta/Elev= 30
    .6961437.453   2.9911437.738   9.5031440.931   10.811441.219  31.0391438.874
  61.3831435.083  71.4971433.637 101.8411428.484 132.1851424.263 152.4141421.102
 162.5281418.938 172.6431415.818 182.7571409.908 202.9861407.973 213.1011404.858
 224.1421402.323 231.3151400.427  233.331399.991 243.4441399.708 253.5591399.833
 263.6741401.311  271.841402.048 273.7881402.245  344.591404.681 415.3911406.029
 445.7351407.833 496.308 1409.84 526.651 1410.15 637.9111414.134 758.5281417.984
#Mann= 3 , 0 , 0
    .696    .035       0 224.142     .07       0  271.84    .035       0
Bank Sta=224.142,271.84
XS Rating Curve= 0 ,0
Exp/Cntr=0.3,0.1

Type RM Length L Ch R = 1 ,57346   ,453.727,498.048,544.871
XS GIS Cut Line= 2
     6258288.506     2213006.936     6258478.324     2213709.609
#Sta/Elev= 30
       01417.151  13.9321417.165  34.6491417.745  54.1021417.075    96.81413.965
 107.1581413.497 126.1161411.841 138.2331409.975 148.592 1408.14 176.4331405.717
 190.0261404.052  235.351402.104 241.8181401.719 249.8311400.675 262.5351398.346
 272.893    1398 283.2521401.588 284.641 1401.65  293.61    1402 355.761    1402
 366.1191402.874 376.478    1404 386.8361402.849 397.1951404.096 459.3451405.887
 500.7791408.096  562.931409.986 614.7221412.915 656.1561415.004  727.861417.425
#Mann= 3 , 0 , 0
       0    .035       0  235.35     .07       0 284.641    .035       0
Bank Sta=235.35,284.641
XS Rating Curve= 0 ,0
Exp/Cntr=0.3,0.1

Type RM Length L Ch R = 1 ,56848   ,463.71,498.764,521.989
XS GIS Cut Line= 2
     6257873.523     2213031.774     6257837.237     2214187.449
#Sta/Elev= 30
       01420.055  28.6261418.347  68.6461414.531  118.671408.131 128.6751406.314
 168.6951405.979   178.7    1404  218.721403.939 368.7941402.031 388.8031400.469
 398.808 1397.56 408.8131396.068 418.8181396.233 428.8231400.354 438.8281402.675
 456.634  1404.3 468.8431405.667 478.8481405.871 498.8581404.232 528.8721404.786
 558.8871404.017 588.9021406.025 640.9411408.031 698.9561408.932 728.9711409.971
  809.01  1411.8 899.055 1413.491029.1191414.4971079.1431416.1851156.2451419.376
#Mann= 3 , 0 , 0
       0    .035       0 368.794     .07       0 456.634    .035       0
Bank Sta=368.794,456.634
XS Rating Curve= 0 ,0
Exp/Cntr=0.3,0.1

Type RM Length L Ch R = 1 ,56349   ,400.121,499.315,547.433
XS GIS Cut Line= 2
     6257421.121     2212990.223     6257314.613     2213552.586
#Sta/Elev= 30
       01423.104  10.3441421.396  30.6991417.563  34.1331416.752  40.8771414.962
  51.0551411.579  59.8041408.971   71.41    1406 122.2991405.874 132.4771404.293
 163.774 1403.07 222.3891402.018 264.7881401.989 274.9661400.875 285.1431396.469
 295.3211394.915 299.4031395.875 315.6771398.866  325.561399.976 366.5661402.039
 397.0991401.872 407.2771402.413 447.9881405.878  487.661410.231 509.0541413.719
  529.411417.814 539.5881419.122 549.7651420.045 559.9431420.492  572.361420.273
#Mann= 3 , 0 , 0
       0    .035       0 264.788     .07       0  325.56    .035       0
Bank Sta=264.788,325.56
XS Rating Curve= 0 ,0
Exp/Cntr=0.3,0.1

Type RM Length L Ch R = 1 ,55849   ,483.814,499.484,509.926
XS GIS Cut Line= 2
     6257079.224     2212801.961     6256792.619     2213246.493
#Sta/Elev= 30
       0 1414.06  76.8651408.335  98.5681406.141 106.7191404.928 117.108    1404
 129.007 1405.48 134.7381405.624 140.9051405.271 152.8031403.954 192.6111402.099
 279.4211399.919 283.6841399.479 286.6551398.555 295.5821394.886 301.1241394.269
  307.48    1394 315.5921394.254 319.3781394.016 328.1731395.117 337.294 1397.93
 344.5281399.609 351.7631399.948 366.9711400.157 402.6661401.956 414.5641403.851
 426.4631406.605 450.2591409.834 481.9771414.847 510.914 1419.07 528.9151420.492
#Mann= 3 , 0 , 0
       0    .035       0 279.421     .07       0 344.528    .035       0
Bank Sta=279.421,344.528
XS Rating Curve= 0 ,0
Exp/Cntr=0.3,0.1

Type RM Length L Ch R = 1 ,55349   ,501.885,500.002,500.816
XS GIS Cut Line= 6
    6256696.5451    2212526.8543    6256569.2877    2212686.6895
    6256477.0868     2212802.494    6256442.5236    2212845.9052
    6256415.5425    2212879.7936    6256339.4156    2212975.4089
#Sta/Elev= 30
       01415.775  17.2971414.488  55.6441410.823  94.5221407.769 106.7741406.453
 198.3221402.198 283.7191399.887   309.11398.262 312.1851397.864 319.3021395.039
 324.074    1394 336.8571394.167 340.6511394.547 347.7671395.967 354.8841398.251
     3621399.962  393.581401.842 400.7691401.692 404.6991401.039 411.8151400.256
 426.0481401.124 440.2811402.591 451.1411404.956 454.8231404.124 472.0451408.331
 481.2171409.876 511.6931410.561 548.7391410.199 561.4911410.748 580.7251411.987
#Mann= 3 , 0 , 0
       0    .035       0   309.1     .07       0     362    .035       0
Bank Sta=309.1,362
XS Rating Curve= 0 ,0
Exp/Cntr=0.3,0.1

Type RM Length L Ch R = 1 ,54849   ,500.709,500,500.43
XS GIS Cut Line= 6
    6256312.2608    2212206.7801    6256102.3601    2212470.4154
      6256015.49    2212579.5241    6255895.5148    2212730.2131
    6255719.0876    2212951.8055    6255642.9384     2213047.449
#Sta/Elev= 30
       01415.891  30.1741413.542  42.9561413.119  68.5211413.318 119.6511411.059
 131.2781409.896 161.9361404.848  221.911400.012  273.041398.025 306.4281397.988
 324.1691396.791 338.538    1394 362.5171394.185 386.702 1398.16 401.7031399.589
 413.6461399.787 458.6341399.662 490.2761400.446 537.312    1400 545.5391400.807
 552.6561400.432 575.6591401.775 587.9821401.965 595.3541401.483 626.7891401.213
 716.2661405.561 812.7481409.2061005.4051412.8111053.5691414.0731083.2011416.215
#Mann= 3 , 0 , 0
       0    .035       0 306.428     .07       0 386.702    .035       0
Bank Sta=306.428,386.702
XS Rating Curve= 0 ,0
Exp/Cntr=0.3,0.1

Type RM Length L Ch R = 1 ,54349   ,487.215,499.118,518.069
XS GIS Cut Line= 2
     6255905.662     2211914.732     6255398.978     2212551.128
#Sta/Elev= 30
       01439.926  38.9591432.791  78.2241427.405 109.4861422.691 119.2331420.214
 128.0391417.192 149.3891408.283 156.5051404.771 160.6161403.172 163.622 1402.52
 170.7381402.021 186.1811401.862 192.0871400.429 199.2041398.077 220.5531396.336
 231.6161396.014  279.78 1395.99  288.441395.497 301.2221393.749 314.0051393.034
 320.1831393.314 326.7871394.013 362.8821396.074 377.1151397.614 390.6991399.915
 434.0471400.005 518.5231402.541 582.4351405.843 633.5651408.014 813.4671418.554
#Mann= 3 , 0 , 0
       0    .035       0  279.78     .07       0 390.699    .035       0
Bank Sta=279.78,390.699
XS Rating Curve= 0 ,0
Exp/Cntr=0.3,0.1
